--- MUDDYCK2.prj (project) ---

Proj Title=MUDDYCK2
Current Plan=p01
Default Exp/Contr=0,0
English Units
Geom File=g01
Flow File=f01
Plan File=p01
BEGIN DESCRIPTION:
END DESCRIPTION:
DSS Export Rating Curves= 0
DSS Export Rating Curve Sorted= 0
DSS Export Volume Flow Curves= 0
DXF OffsetX= 0
DXF OffsetY= 0
DXF ScaleX= 0
DXF ScaleY= 0

--- MUDDYCK2.p01 (plan) ---

Plan Title=Floodplain
Program Version=4.00
Geom File=g01
Flow File=f01
K Sum by GR=0
Std Step Tol=0.01
Critical Tol=0.01
Num of Std Step Trials=20
Max Error Tol=0.3
Flow Tol Ratio=0.001
Split Flow NTrial=30
Split Flow Tol=0.02
Split Flow Ratio=0.02
Log Output Level=0
Friction Slope Method=1
Unsteady Friction Slope Method=2
Unsteady Bridges Friction Slope Method=1
Global Log Level=0
CheckData=False
Run HTab=0
Run UNet=0
Run PostProcess=0
UNET Theta=0
UNET Theta Warmup=0
UNET ZTol=0
UNET ZSATol=0
UNET MxIter=0
UNET MaxInSteps=0
UNET DtIC=0
UNET DtMin=0
UNET MaxCRTS=0
UNET WFStab=0
UNET SFStab=0
UNET WFX=0
UNET SFX=0
UNET DSS MLevel=0
UNET DZMax Abort=0
UNET Convert EG Bridges=0
UNET Use Existing IB Tables=0
UNET Froude Limit=0
UNET Froude Power=0
Write IC File=0
Echo Input=False
Echo Output=False
Write Detailed=0

--- MUDDYCK2.f01 (steady flow) ---

Flow Title=NFF Regression Equation
Program Version=4.10
Number of Profiles= 1
Profile Names=P100yr
River Rch & RM=MUDDYCK2,Main            ,61006.5
709.4375
River Rch & RM=MUDDYCK2,Main            ,59116.1
720.1426
River Rch & RM=MUDDYCK2,Main            ,58672.7
780.1704
River Rch & RM=MUDDYCK2,Main            ,56355.5
830.0394
River Rch & RM=MUDDYCK2,Main            ,53174.4
 886.498
River Rch & RM=MUDDYCK2,Main            ,52506
1074.594
River Rch & RM=MUDDYCK2,Main            ,49816.2
1131.235
River Rch & RM=MUDDYCK2,Main            ,47227.8
 1180.56
River Rch & RM=MUDDYCK2,Main            ,46479.3
1231.543
River Rch & RM=MUDDYCK2,Main            ,44141.2
1254.992
River Rch & RM=MUDDYCK2,Main            ,42803.8
1524.654
River Rch & RM=MUDDYCK2,Main            ,41786.3
1694.625
River Rch & RM=MUDDYCK2,Main            ,40689.9
1860.558
River Rch & RM=MUDDYCK2,Main            ,36256.8
1935.128
River Rch & RM=MUDDYCK2,Main            ,35231.8
2372.151
River Rch & RM=MUDDYCK2,Main            ,32995.7
2395.018
River Rch & RM=MUDDYCK2,Main            ,25557.6
2515.685
River Rch & RM=MUDDYCK2,Main            ,20305.9
2674.353
River Rch & RM=MUDDYCK2,Main            ,16202.3
 2828.08
River Rch & RM=MUDDYCK2,Main            ,11813.1
2983.257
River Rch & RM=MUDDYCK2,Main            ,622.1
3194.336
Boundary for River Rch & Prof#=MUDDYCK2,Main            , 1
Up Type= 0
Dn Type= 1
Dn Known WS=1475.3
DSS Import GetInterval= 0
DSS Import GetPeak= 0
DSS Import FillOption= 0

--- MUDDYCK2.g01 (geometry) ---

Geom Title=USGS 10m DEM
Program Version=4.10

River Reach=MUDDYCK2        ,Main
Reach XY= 30
     1960835.079      383259.668     1960232.351      384092.076
     1960563.466      385435.252     1959175.661      387030.724
     1960167.208       390641.68     1956858.934      393919.001
     1956281.282      394870.238     1956412.273      396558.461
     1953725.611      396766.044      1951754.07      395407.203
     1948543.331      395450.014     1947740.101      394474.871
     1946308.076      394902.003     1946476.279      396670.817
     1945897.124      396762.564     1943533.584      394252.689
     1942635.147      394441.491     1940459.944      396556.515
     1939427.021      395625.661      1939493.92      394104.184
     1938384.541      393483.742     1938800.021      391206.343
     1936864.593      389955.672     1936463.963      388604.309
     1932384.644      385593.848     1932331.125      384367.874
      1931597.82      383744.876      1931908.15      383245.744
     1931302.357      382890.944     1931672.364      382105.625

Type RM Length L Ch R = 1 ,61006.5 ,225.9,215.9,205.3
XS GIS Cut Line= 2
     1960728.655      383130.066     1960926.572      383398.295
#Sta/Elev= 24
       0  2402.4     9.8 2401.12    19.6 2399.95      49 2396.92    78.4 2394.26
   107.8 2391.88   117.6 2390.98   127.4 2389.95   137.3 2389.14   147.1 2389.06
   156.9 2389.75   166.7 2390.67   176.5 2391.31   186.3 2391.66   196.1 2391.88
   205.9 2391.85   215.7 2391.56   225.5 2391.14   235.3 2390.93   245.1  2391.3
   254.9 2392.32   294.1 2397.39   323.5 2401.08   333.3 2402.21
#Mann= 3 , 0 , 0
       0      .1       0   127.4    .045       0   166.7      .1       0
#XS Ineff= 2 , 0
                          197.18         2391.88
Permanent Ineff=
       F       F
Bank Sta=127.4,166.7
XS Rating Curve= 0 ,0
Exp/Cntr=0.3,0.1

Type RM Length L Ch R = 1 ,60790.6 ,181.3,189.5,197.8
XS GIS Cut Line= 2
     1960624.489      383369.649     1960840.635      383497.253
#Sta/Elev= 29
       0 2392.87     9.6 2391.94    19.3  2391.1      29 2390.48    38.6 2390.11
    48.3 2389.81    57.9 2389.55    67.6 2389.22    77.2 2388.92    86.9 2388.53
    96.5 2387.81   106.2 2385.98   114.4 2383.88   115.8 2383.52   125.5 2382.28
   129.4 2382.82   135.2 2383.62   144.8  2387.7   154.5 2392.02   164.1 2394.27
   173.8  2395.1   183.4 2395.59   193.1    2396   202.7 2396.36   212.4 2396.85
     222 2397.47   231.7 2398.32   241.4 2399.27     251 2400.41
#Mann= 3 , 0 , 0
       0     .06       0   114.4    .045       0   135.2     .06       0
Bank Sta=114.4,135.2
XS Rating Curve= 0 ,0
Exp/Cntr=0.3,0.1

Type RM Length L Ch R = 1 ,60601.1 ,132.6,135.5,137.8
XS GIS Cut Line= 2
      1960543.76      383489.441      1960668.76      383640.482
#Sta/Elev= 23
       0 2387.28     9.8 2387.41    19.6 2387.62    29.4 2387.83    39.2  2387.7
      49  2387.4    58.8 2387.08    68.6  2386.8    78.4 2386.36    88.2 2385.38
      98 2383.76   107.8 2381.53   117.6 2379.73   122.5 2379.85   127.4 2379.97
   137.2 2383.14   137.5 2383.32     147 2388.91   156.8 2393.43   166.6 2395.28
   176.4 2396.34   186.2 2397.23   196.1 2397.93
#Mann= 3 , 0 , 0
       0     .06       0   107.8    .045       0   137.5     .06       0
Bank Sta=107.8,137.5
XS Rating Curve= 0 ,0
Exp/Cntr=0.3,0.1

Type RM Length L Ch R = 1 ,60465.6 ,38.5,38.5,38.5
XS GIS Cut Line= 2
     1960438.725      383548.468     1960560.253      383732.496
#Sta/Elev= 26
       0 2385.68     9.6 2384.83    19.2 2384.01    28.8 2383.24    38.4 2383.33
    47.9 2384.12    57.5  2385.8    67.1 2386.87    76.7 2387.44    86.3 2387.31
    95.9 2386.85   105.5 2386.39   115.1  2385.5   124.6  2383.4   129.1  2381.9
   134.2 2380.21   143.8  2378.8   144.1 2378.91   153.4 2382.28     163 2385.88
   172.6 2388.01   182.2 2389.01   191.8 2389.98   201.4 2390.99     211 2392.04
   220.5 2393.12
#Mann= 3 , 0 , 0
       0     .06       0   129.1    .045       0   153.4     .06       0
#XS Ineff= 2 , 0
           76.41  2387.5
Permanent Ineff=
       F       F
Bank Sta=129.1,153.4
XS Rating Curve= 0 ,0
Exp/Cntr=0.3,0.1

Type RM Length L Ch R = 1 ,60427.1 ,258.7,249.5,240.1
XS GIS Cut Line= 2
     1960410.079       383574.51     1960531.607      383758.538
#Sta/Elev= 26
       0  2391.5     9.6 2390.66    19.2 2389.74    28.8 2388.74    38.4 2387.78
    47.9 2386.83    57.5 2386.07    67.1 2385.48    76.7    2385    86.3 2384.63
    95.9 2384.36   105.5 2384.14   115.1 2383.14   119.8 2381.42   124.6 2379.66
   134.2 2376.79   134.8 2376.88   143.8 2378.29   153.4 2381.37     163    2384
   172.6 2385.62   182.2  2386.7   191.8 2387.65   201.4 2388.52     211 2389.34
   220.5 2390.15
#Mann= 3 , 0 , 0
       0     .06       0   124.6    .045       0   143.8     .06       0
Bank Sta=124.6,143.8
XS Rating Curve= 0 ,0
Exp/Cntr=0.3,0.1

Type RM Length L Ch R = 1 ,60177.6 ,592.1,573.8,551.5
XS GIS Cut Line= 2
     1960212.162      383796.732     1960410.079      383925.205
#Sta/Elev= 27
       0  2411.3     9.8 2409.03    19.7 2406.75    29.5 2404.09    39.3 2400.76
    49.2 2396.57      59 2391.82    68.8 2386.31    78.6 2380.92    88.5 2375.97
    98.3 2371.98   108.2 2369.15   115.7 2368.51     118 2368.31   127.8 2368.54
   130.7 2368.93   137.6 2369.86   147.5 2371.76   157.3  2373.5   167.1 2374.95
     177 2375.84   186.8  2376.1   196.6 2376.04   206.5 2376.07   216.3 2376.27
   226.1 2376.54     236 2376.81
#Mann= 3 , 0 , 0
       0      .1       0   115.7    .045       0   130.7     .06       0
Bank Sta=115.7,130.7
XS Rating Curve= 0 ,0
Exp/Cntr=0.3,0.1

Type RM Length L Ch R = 1 ,59603.9 ,483.9,487.8,491.5
XS GIS Cut Line= 2
     1960201.746      384442.566      1960552.44       384324.51
#Sta/Elev= 27
       0 2397.82     9.7 2395.07    19.5 2391.87    29.2 2388.45      39 2385.18
    58.4 2378.97    68.2 2375.19    77.9 2370.79    87.6 2365.55    97.4 2358.62
   107.1  2352.4   108.7 2352.12   116.8 2350.71   123.7 2352.99   126.6 2353.95
   136.3 2358.03   146.1 2359.86   155.8 2360.37   194.8 2361.65   204.5 2362.24
   214.2 2363.24   243.4 2366.86   272.7 2370.29   321.3 2375.75   331.1 2376.76
   350.6 2378.58     370 2380.17
#Mann= 3 , 0 , 0
       0      .1       0   108.7    .045       0   123.7      .1       0
Bank Sta=108.7,123.7
XS Rating Curve= 0 ,0
Exp/Cntr=0.3,0.1

Type RM Length L Ch R = 1 ,59116.1 ,437,443.4,449.6
XS GIS Cut Line= 2
      1960431.78      384846.211     1960642.718      384809.753
#Sta/Elev= 25
       0 2355.95     9.7 2354.76    19.5 2353.53    29.2 2352.36    38.9 2351.37
    48.6 2350.81    58.4 2350.64    68.1  2350.6    77.8 2350.34    87.6 2349.31
    89.3 2348.95    97.3 2347.26   104.3 2346.03     107 2345.56   116.8 2345.39
   126.5 2347.14   136.2 2351.84     146 2357.74   155.7 2359.83   165.4 2360.35
   175.1 2360.82   184.9 2361.23   194.6 2361.62   204.3 2361.89   214.1 2362.26
#Mann= 3 , 0 , 0
       0     .06       0    89.3    .045       0   126.5     .06       0
Bank Sta=89.3,126.5
XS Rating Curve= 0 ,0
Exp/Cntr=0.3,0.1

Type RM Length L Ch R = 1 ,58672.7 ,333,336.7,340.3
XS GIS Cut Line= 2
     1960228.655      385244.649     1960948.273      385279.371
#Sta/Elev= 30
       0  2345.2    38.9 2344.62    68.2 2343.79   107.1 2342.86     146 2342.32
   253.1 2341.14     331 2341.66   351.1 2341.47   360.2 2341.43   366.1 2341.65
     370 2341.79   379.7 2342.54   389.4 2343.46   408.9 2345.08   418.6 2346.03
   428.4 2347.36   447.8 2350.75   467.3 2354.01   486.8 2357.03   506.3  2359.8
   525.7 2362.72   545.2 2365.84   584.2 2372.54   593.9 2374.11   613.4 2376.91
   632.8 2379.91   652.3 2382.69     662  2383.9   691.2 2387.05   720.5 2390.91
#Mann= 3 , 0 , 0
       0     .06       0   351.1    .045       0   366.1     .06       0
Bank Sta=351.1,366.1
XS Rating Curve= 0 ,0
Exp/Cntr=0.3,0.1

Type RM Length L Ch R = 1 ,58335.9 ,494.4,516.8,537
XS GIS Cut Line= 3
     1960160.554      385380.131     1960267.325      385502.526
     1960676.179      385614.506
#Sta/Elev= 30
       0 2339.95    57.3 2336.99   143.3 2334.83   152.9 2334.22   162.4 2333.35
   172.1 2333.01   181.7 2332.94   191.3 2333.18     201 2333.71   229.9 2335.99
   239.5 2336.55   249.1 2336.85     278  2337.3   297.3 2337.12   355.1 2335.24
   364.7 2334.67   373.1 2333.81     384 2333.14   388.1 2333.72   393.6  2334.5
   412.9  2340.3   422.6 2342.31   432.2  2343.4   451.4 2344.88   461.1 2346.01
   470.7 2347.64   480.4 2349.68   499.6 2354.08   518.9 2357.02   586.3 2370.08
#Mann= 3 , 0 , 0
       0     .06       0   373.1    .045       0   388.1     .06       0
#XS Ineff= 2 , 0
          278.03  2337.5
Permanent Ineff=
       F       F
Bank Sta=373.1,388.1
XS Rating Curve= 0 ,0
Exp/Cntr=0.3,0.1

Type RM Length L Ch R = 1 ,57819.2 ,870.1,871.5,868.6
XS GIS Cut Line= 3
     1960090.635      385532.843     1960222.579      385942.566
     1960285.079       386012.01
#Sta/Elev= 30
       0 2335.99     9.8 2336.18    19.6 2335.95    29.4 2334.48    39.1 2332.19
    48.9 2331.35   107.6 2331.33   156.5 2330.75   176.1 2330.35   185.9 2329.82
   195.7 2328.92   205.4 2327.74   215.2  2326.4     225 2324.86   234.8 2323.83
   254.4 2323.78   264.1 2323.84   322.8 2324.42     362 2324.52   371.8 2324.68
   381.5 2325.19   391.3 2326.05   420.7 2328.98   430.4 2330.63   439.8 2333.82
   449.1  2338.2   458.5 2342.78   467.8 2346.85   477.2 2350.22   523.9 2365.94
#Mann= 3 , 0 , 0
       0     .06       0   234.8    .045       0   264.1      .1       0
Bank Sta=234.8,264.1
XS Rating Curve= 0 ,0
Exp/Cntr=0.3,0.1

Type RM Length L Ch R = 1 ,56947.6 ,616.4,592.1,566.4
XS GIS Cut Line= 2
     1959382.301       385855.76     1959649.662      386432.149
#Sta/Elev= 30
       0 2329.84    39.1 2328.74    97.8 2324.46   156.4 2320.77   166.2  2320.3
   185.7 2320.14   195.5 2320.39   205.3    2321   234.6 2323.74   244.4 2324.26
   254.2 2324.38   293.2 2322.93   312.8 2323.31   332.4    2324   342.1 2323.57
   351.9 2322.48   371.4 2319.51     391 2316.76   469.2 2306.44     479 2305.66
   488.8 2305.81   494.7 2307.02   498.5  2307.8   527.8 2317.79   557.2 2330.28
   586.5 2340.98   596.3 2344.08     606 2346.92   625.6  2352.2   635.4 2354.56
#Mann= 3 , 0 , 0
       0     .06       0   469.2    .045       0   494.7      .1       0
Bank Sta=469.2,494.7
XS Rating Curve= 0 ,0
Exp/Cntr=0.3,0.1

Type RM Length L Ch R = 1 ,56355.5 ,528.3,526.9,517.3
XS GIS Cut Line= 3
     1959058.991      386726.485     1959327.221      386723.881
     1959460.033      386757.735
#Sta/Elev= 26
       0 2311.24    19.2  2309.9    47.9 2307.74    57.5 2307.11    76.6 2306.06
    86.2 2305.68   162.9 2303.11   172.4 2302.72   210.8 2300.69   229.9 2299.83
   249.1 2299.15   258.7 2299.48   268.2 2301.37     278 2304.88   287.8  2308.6
   297.6 2312.17   307.4 2316.54   317.2 2321.48     327 2326.59   336.8 2331.81
   346.6 2337.15   356.4 2342.67   375.9  2354.2   385.7 2359.69   395.5 2364.24
   405.3 2368.27
#Mann= 3 , 0 , 0
       0      .1       0   229.9    .045       0   258.7      .1       0
Bank Sta=229.9,258.7
XS Rating Curve= 0 ,0
Exp/Cntr=0.3,0.1

Type RM Length L Ch R = 1 ,55828.7 ,706.8,705.2,703.6
XS GIS Cut Line= 2
     1959010.773      387189.093     1959385.773      387192.566
#Sta/Elev= 30
       0 2301.37    19.2 2301.88    28.8 2301.94    48.1 2301.39    57.7 2300.58
    67.3 2299.36    96.2 2294.88   105.8 2293.88     125 2293.19   144.2 2293.32
   153.8 2293.15   163.5 2292.24   173.1 2290.81   182.7 2290.16   192.3  2290.5
   240.4 2296.48     250 2299.59   259.6 2305.78   269.2 2312.76   278.9  2318.7
   288.5 2324.14   298.1 2329.32   307.7 2333.93   317.3 2338.03   326.9 2341.61
   336.6 2344.43   346.2 2346.74   355.8 2349.42   365.4 2352.91     375 2356.69
#Mann= 3 , 0 , 0
       0      .1       0   173.1    .045       0   192.3      .1       0
Bank Sta=173.1,192.3
XS Rating Curve= 0 ,0
Exp/Cntr=0.3,0.1

Type RM Length L Ch R = 1 ,55123.4 ,897.3,890.8,884.1
XS GIS Cut Line= 3
     1959253.829      387834.927     1959503.829      387817.566
     1959604.523      387768.955
#Sta/Elev= 26
       0 2292.62    19.3 2291.92    86.8 2289.93   134.9  2288.1   154.2 2286.96
   163.9 2286.24   173.5 2284.48   183.1 2280.78   192.8 2277.22   202.4 2275.85
     212 2276.57   214.7 2277.21   221.7 2278.88   231.3 2281.85   250.6 2287.41
   259.9 2290.84   269.2 2295.46   278.6  2301.2   287.9 2307.03   306.5  2318.3
   315.8  2323.8   325.1 2328.92   334.5 2333.62   343.8 2337.75   353.1 2341.24
   362.4 2344.25
#Mann= 3 , 0 , 0
       0      .1       0   192.8    .045       0   214.7      .1       0
Bank Sta=192.8,214.7
XS Rating Curve= 0 ,0
Exp/Cntr=0.3,0.1

Type RM Length L Ch R = 1 ,54232.6 ,685.2,683.1,674.9
XS GIS Cut Line= 2
     1959528.135      388734.232      1959958.69      388571.038
#Sta/Elev= 30
       0 2296.33    19.6 2289.29      49 2278.37    58.8 2275.57    68.6 2274.28
    78.4 2274.22    88.2 2274.64   127.4 2277.67     147 2279.02   156.8 2279.51
   166.5 2279.42   176.3 2278.71   215.5  2274.9   235.1 2272.83   254.7 2270.49
   264.5 2268.96   274.3 2267.37   284.1 2267.15   293.9 2269.72   303.7 2275.13
   313.5 2281.49   323.3 2287.38   372.3 2315.61   382.1  2320.9   391.9 2325.51
   401.7 2329.58   411.5  2333.2   431.1 2339.43   450.6 2345.16   460.4 2348.52
#Mann= 3 , 0 , 0
       0     .06       0   264.5    .045       0   293.9      .1       0
Bank Sta=264.5,293.9
XS Rating Curve= 0 ,0
Exp/Cntr=0.3,0.1

Type RM Length L Ch R = 1 ,53549.5 ,363,375.1,392.4
XS GIS Cut Line= 3
     1959788.551      389369.649     1960163.551      389185.621
     1960354.523      389029.371
#Sta/Elev= 30
       0 2296.04    38.9 2281.63      68 2270.34    77.7 2267.19    87.4 2265.14
    97.1 2264.37   126.3 2264.09   174.9 2264.69   223.4 2265.74   242.9 2265.85
   262.3 2265.27   310.9 2263.24   351.8 2262.34   378.9 2261.71   388.6 2262.67
     408 2265.54   417.7  2267.6   427.2 2270.43   436.7 2274.17   446.2 2278.75
   465.2 2288.39   474.7 2292.87   484.2 2297.05   512.6 2309.05   531.6 2316.27
   550.6 2322.71   560.1 2325.55     598 2336.21     636 2347.39   664.5 2356.75
#Mann= 3 , 0 , 0
       0      .1       0   351.8    .045       0   388.6     .06       0
#XS Ineff= 2 , 0
          233.66 2266.34
Permanent Ineff=
       F       F
Bank Sta=351.8,388.6
XS Rating Curve= 0 ,0
Exp/Cntr=0.3,0.1

Type RM Length L Ch R = 1 ,53174.4 ,668.6,668.4,461.4
XS GIS Cut Line= 3
     1959868.412      389595.343     1959993.412      389546.732
      1960396.19      389557.149
#Sta/Elev= 30
       0 2315.88    47.9 2302.13    67.1 2296.38    76.6 2293.22    86.2 2289.37
    95.8 2284.66     115 2274.58   124.5 2270.11     144 2261.98   153.8 2259.49
   163.6 2259.04   183.3 2259.36   242.2 2261.32   271.7 2260.56   320.8 2258.14
   330.7 2257.84   340.5 2257.94  349.862258.819     370 2262.04   389.6 2264.36
   399.4 2264.72   448.6 2264.85   458.4 2265.19   468.2 2266.41   478.1  2268.7
   497.7 2274.14   507.6 2276.52   517.4  2278.5   527.2 2280.07     537 2281.18
#Mann= 3 , 0 , 0
       0      .1       0   320.8    .045       0  349.86      .1       0
#XS Ineff= 2 , 0
          243.38 2261.57
Permanent Ineff=
       F       F
Bank Sta=320.8,349.86
XS Rating Curve= 0 ,0
Exp/Cntr=0.3,0.1

Type RM Length L Ch R = 1 ,52506   ,314.5,305.1,295.6
XS GIS Cut Line= 2
     1959875.357      389866.177     1960354.523       389887.01
#Sta/Elev= 30
       0 2291.13    29.4 2281.34    39.2 2278.38    48.9 2275.96    68.5  2272.5
    97.9 2270.22   107.7 2268.96   117.5 2266.97   127.2 2264.15   146.8 2255.26
   156.6  2252.2   166.4 2250.59   176.2 2249.46     186 2249.48   195.8 2251.18
   215.3 2255.62   225.1    2257   234.9 2257.84   342.6 2260.91   352.4 2261.87
   362.2 2264.37     372 2267.79   401.3 2279.08   411.1 2280.94   420.9 2282.08
   430.7 2284.74   450.2 2293.51     460 2297.14   469.8 2299.53   479.6 2300.99
#Mann= 3 , 0 , 0
       0      .1       0   166.4    .045       0   195.8      .1       0
Bank Sta=166.4,195.8
XS Rating Curve= 0 ,0
Exp/Cntr=0.3,0.1

Type RM Length L Ch R = 1 ,52200.9 ,508.7,521.6,534.4
XS GIS Cut Line= 2
      1959918.76      390231.628      1960271.19      390109.232
#Sta/Elev= 30
       0 2264.75     9.8 2262.75    19.6    2261    29.4 2259.73    39.3 2259.08
    58.9 2258.45    98.2  2256.6     108 2256.24   117.8 2256.08   137.4 2256.34
   147.3 2256.14   166.9 2255.47   176.7 2255.23   186.5 2255.05   206.2 2255.06
     216 2254.56   225.8 2252.43   235.6    2249   245.4  2249.3   249.4 2251.05
   255.3 2253.63   265.1 2257.31   274.9 2258.78   304.4 2260.05   314.2 2260.82
     324 2261.87   333.8 2263.59   343.6 2266.57   353.4 2270.57   373.1 2279.25
#Mann= 3 , 0 , 0
       0      .1       0   225.8    .045       0   249.4      .1       0
Bank Sta=225.8,249.4
XS Rating Curve= 0 ,0
Exp/Cntr=0.3,0.1

Type RM Length L Ch R = 1 ,51679.3 ,879.2,880,880.5
XS GIS Cut Line= 2
     1959875.357      390588.399     1960351.051      390706.455
#Sta/Elev= 30
       0    2277     9.8  2272.4    19.6 2268.53    29.4  2264.9      49 2256.45
    58.8 2252.93    68.6 2250.72    78.4 2250.07     147 2250.11   205.8 2249.83
   254.9 2248.85   264.7 2248.22   274.5 2246.78   284.3 2244.68   294.1 2243.36
   301.9 2244.74   303.9  2245.1   313.7 2252.41   323.5 2262.64   333.3 2270.59
   343.1 2277.25   362.7 2289.57   372.5 2295.91   382.3 2301.86   411.7 2318.66
   421.5 2324.09   450.9  2339.6   460.7 2344.22   470.5 2348.28   490.1 2355.98
#Mann= 3 , 0 , 0
       0      .1       0   284.3    .045       0   301.9      .1       0
Bank Sta=284.3,301.9
XS Rating Curve= 0 ,0
Exp/Cntr=0.3,0.1

Type RM Length L Ch R = 1 ,50799.3 ,492.1,500.8,509.7
XS GIS Cut Line= 3
     1959455.218       391262.01     1959760.773      391352.288
     1959840.635      391439.093
#Sta/Elev= 30
       0  2313.9     9.6 2308.79    19.3 2302.49      29 2294.03    38.6 2284.43
    48.3 2275.15    57.9 2267.74    67.6 2262.81   106.2 2245.07   135.2  2235.1
   144.8 2233.55   154.5  2233.5   164.1 2234.94   173.8 2237.26   183.4 2238.53
   202.8 2238.64   212.4 2239.48   231.7 2241.98     251 2243.92   299.3 2246.43
     309 2247.61   318.6  2249.5   328.4  2252.3   338.3 2255.83   348.1 2260.24
   357.9 2265.29   367.8 2270.68   397.2  2289.1   426.7 2306.38   436.6 2311.72
#Mann= 3 , 0 , 0
       0      .1       0   135.2    .045       0   173.8      .1       0
Bank Sta=135.2,173.8
XS Rating Curve= 0 ,0
Exp/Cntr=0.3,0.1

Type RM Length L Ch R = 1 ,50298.5 ,480.9,482.3,483.7
XS GIS Cut Line= 2
     1959262.116      391640.547       1959501.7      391833.256
#Sta/Elev= 27
       0 2287.27    19.2 2277.34    28.8 2272.53    38.4 2267.95      48 2263.78
    57.6 2259.83    67.3 2256.11    76.9 2252.56    86.5 2249.57   115.3  2242.1
   124.9 2239.82     1372237.251   144.1 2235.72   153.7 2233.45   163.3 2231.75
   166.42231.634     173 2231.38   182.6 2233.08   192.2 2236.12   201.8 2239.33
   211.4 2242.97     221 2247.94   230.6 2254.12   240.2 2260.12   249.8 2264.84
   278.6 2277.14   307.5 2289.71
#Mann= 3 , 0 , 0
       0      .1       0     137    .045       0   166.4      .1       0
Bank Sta=137,166.4
XS Rating Curve= 0 ,0
Exp/Cntr=0.3,0.1

Type RM Length L Ch R = 1 ,49816.2 ,654.4,657.2,659.7
XS GIS Cut Line= 3
     1958930.912      391914.788     1959014.246      392050.205
     1959198.273      392216.871
#Sta/Elev= 30
       0 2289.37     9.4 2286.46    28.1 2280.44    56.1 2271.23    84.2 2261.82
    93.5 2258.53   112.2 2251.53   121.6 2248.29   130.9 2245.77   140.3 2243.96
   149.6 2242.51   168.6 2239.77   197.2 2235.48   206.8 2234.12   225.8 2231.66
   235.4 2230.28     245 2228.99   254.5 2228.42     264 2229.51   273.6 2231.33
   283.1 2233.31   302.2 2236.51   311.8  2238.6   321.3 2242.32   330.9 2247.59
   359.5 2264.76   378.6  2275.8   388.2 2281.08   397.7  2285.8   407.3 2290.17
#Mann= 3 , 0 , 0
       0      .1       0   235.4    .045       0     264      .1       0
Bank Sta=235.4,264
XS Rating Curve= 0 ,0
Exp/Cntr=0.3,0.1

Type RM Length L Ch R = 1 ,49159   ,415.1,405.8,396.4
XS GIS Cut Line= 2
     1958465.241      392328.047     1958673.575      392572.839
#Sta/Elev= 24
       0 2258.41    29.2 2246.75    58.4 2235.31    68.2  2232.1    77.9 2230.21
   116.9 2224.78   126.6 2223.59   146.1 2221.61   155.8 2220.34   165.6 2219.26
   175.3 2219.34   185.1 2221.48  185.35 2221.59   204.6 2230.15   214.3 2234.24
     224 2238.58   233.8 2242.58   243.5 2246.33   253.3 2249.98   282.5 2260.12
   292.2 2263.35     302 2266.15   311.7 2268.16   321.4 2269.81
#Mann= 3 , 0 , 0
       0      .1       0   146.1    .045       0  185.35      .1       0
Bank Sta=146.1,185.35
XS Rating Curve= 0 ,0
Exp/Cntr=0.3,0.1

Type RM Length L Ch R = 1 ,48753.2 ,618.5,629.7,640.6
XS GIS Cut Line= 3
     1958156.607      392650.899     1958278.135      392737.705
     1958455.218       392824.51
#Sta/Elev= 27
       0 2275.43      28 2263.83    37.3 2260.06    46.7 2256.53      56 2253.21
    74.7 2246.84   102.7 2237.14   121.3  2230.5   130.7 2227.26     140  2224.2
   149.4 2221.32   158.7 2218.04   168.1 2214.24   177.5  2210.9     181 2210.29
   186.9 2209.27     196 2210.02   205.7 2212.05   215.1 2214.26   224.5 2216.28
     262 2223.72   271.4 2225.66   280.8 2228.07   290.2 2231.01   299.6  2234.2
     309 2237.53   346.6 2251.24
#Mann= 3 , 0 , 0
       0      .1       0     181    .045       0     196      .1       0
Bank Sta=181,196
XS Rating Curve= 0 ,0
Exp/Cntr=0.3,0.1

Type RM Length L Ch R = 1 ,48123.5 ,897.2,895.7,894.2
XS GIS Cut Line= 2
     1957774.662      393060.621      1957958.69      393314.093
#Sta/Elev= 27
       0 2247.32    29.4  2236.5    39.2 2232.96    48.9 2229.52    58.7 2226.24
    68.5 2223.14   107.7 2211.32   117.5 2208.26   127.2  2204.7     137 2201.61
   139.82201.296   146.8 2200.51   154.82201.432   156.6 2201.64   166.4  2204.2
   176.2 2206.62   195.8 2210.84   205.6 2213.28   215.4  2216.6   225.1 2220.66
   234.9  2225.2   264.3 2239.73   274.1 2244.38   283.9 2248.83   293.7 2253.11
   303.4 2257.23   313.2 2261.14
#Mann= 3 , 0 , 0
       0      .1       0   139.8    .045       0   154.8      .1       0
Bank Sta=139.8,154.8
XS Rating Curve= 0 ,0
Exp/Cntr=0.3,0.1

Type RM Length L Ch R = 1 ,47227.8 ,491.2,472,452.8
XS GIS Cut Line= 2
     1957010.773      393536.316     1957201.746      393768.955
#Sta/Elev= 19
       0 2234.53    19.4 2228.31    48.6  2218.6    77.7 2208.48   116.5 2194.55
   126.2 2191.38   135.9 2189.13   145.6 2188.04   174.8 2185.57   184.5 2184.95
   194.2 2185.08   203.9 2185.97   213.6 2187.55   223.3 2189.33     233 2191.18
   252.4 2195.12   271.9 2198.88   291.3 2202.34     301 2203.87
#Mann= 3 , 0 , 0
       0      .1       0   174.8    .045       0   203.9      .1       0
Bank Sta=174.8,203.9
XS Rating Curve= 0 ,0
Exp/Cntr=0.3,0.1

Type RM Length L Ch R = 1 ,46755.8 ,260.5,276.5,291.2
XS GIS Cut Line= 3
     1956611.468      393973.816     1956722.579      394022.427
     1956986.468      394032.843
#Sta/Elev= 30
       0 2239.05     9.3 2234.06    18.7 2229.17      28 2224.49    37.3 2220.04
    46.6 2215.92      56 2212.38    65.3  2209.3      84 2203.72    93.3 2200.64
   102.6 2196.73     112 2191.32   121.3 2185.31   131.1 2180.68   140.8 2178.69
   189.8 2175.06   209.3  2173.5   219.1 2172.57   228.9 2171.62   238.6 2171.35
   247.8  2172.5   248.4 2172.57   258.2 2174.85     268 2176.92   277.8 2178.32
   287.6 2179.32   297.3 2180.13   316.9 2181.37     356 2183.31   385.4 2184.65
#Mann= 3 , 0 , 0
       0      .1       0   219.1    .045       0   247.8      .1       0
Bank Sta=219.1,247.8
XS Rating Curve= 0 ,0
Exp/Cntr=0.3,0.1

Type RM Length L Ch R = 1 ,46479.3 ,220.3,228.4,236
XS GIS Cut Line= 2
     1956746.885      394216.871     1956930.912      394362.705
#Sta/Elev= 27
       0 2186.11     9.8 2182.95    19.6 2179.62    29.4 2176.15    39.1 2172.95
    48.9 2170.68    58.7  2169.8    68.5 2169.44    78.3 2169.08      88 2168.73
    97.8 2168.38   107.6 2167.83   112.8 2167.38   117.4 2166.98   127.2 2166.15
   127.8 2166.19     137 2166.77   146.8 2170.06   156.5  2174.3   166.3 2178.02
   176.1 2181.52   185.9  2185.3   195.7 2189.24   205.4 2193.19   215.2 2197.13
     225 2200.97   234.8 2204.81
#Mann= 3 , 0 , 0
       0      .1       0   112.8    .045       0   146.8      .1       0
Bank Sta=112.8,146.8
XS Rating Curve= 0 ,0
Exp/Cntr=0.3,0.1

Type RM Length L Ch R = 1 ,46250.9 ,300.1,281.9,264.1
XS GIS Cut Line= 3
     1956587.162      394303.677     1956673.968      394446.038
     1956726.051      394505.066
#Sta/Elev= 28
       0  2189.8     9.8 2188.67    19.6  2187.5    29.4 2186.34    39.2 2185.11
      49 2183.87    58.8 2182.29    68.7  2178.9    78.5 2173.15    88.3 2166.76
    98.1  2162.9   107.9 2161.35   117.7 2160.25   127.5  2159.1   137.3 2157.95
   139.8 2157.75   147.1 2157.18   154.8 2157.42   156.9 2157.48   166.7 2159.81
   176.6 2162.97   186.4 2165.82   196.3  2168.5   206.1 2171.27   215.9 2174.04
   225.8 2176.96   235.6 2180.04   245.5 2183.22
#Mann= 3 , 0 , 0
       0      .1       0   137.3    .045       0   156.9      .1       0
Bank Sta=137.3,156.9
XS Rating Curve= 0 ,0
Exp/Cntr=0.3,0.1

Type RM Length L Ch R = 1 ,45969   ,596.2,584.9,572.9
XS GIS Cut Line= 3
     1956218.239      394481.628     1956436.989      394627.461
     1956798.968      394718.607
#Sta/Elev= 30
       0 2238.96     9.7 2232.98    19.5 2228.06    77.9 2200.98    87.6 2197.14
    97.4 2194.26   146.1 2181.61   165.5 2177.34     185 2174.16   194.7 2172.87
   233.7 2168.98   243.4 2167.19   253.2 2164.32   272.7 2157.38   282.6 2154.57
   292.4 2153.51   321.8 2154.19   331.7 2153.83   361.1 2151.42     371 2150.53
   380.8 2150.43   390.6 2152.22   420.1 2162.98   469.2 2178.09   488.8 2185.19
   498.7 2189.34     538 2206.39   557.6 2215.95   587.1 2231.18   636.2 2258.32
#Mann= 3 , 0 , 0
       0      .1       0   361.1    .045       0   390.6      .1       0
Bank Sta=361.1,390.6
XS Rating Curve= 0 ,0
Exp/Cntr=0.3,0.1

Type RM Length L Ch R = 1 ,45384.1 ,366.3,376.5,386.5
XS GIS Cut Line= 2
      1956208.69      395046.732     1956399.662      395001.593
#Sta/Elev= 23
       0 2148.16     9.8  2146.7    19.6 2145.22    29.4 2143.74    39.2 2142.25
    49.1 2140.83    58.9 2139.32    68.7 2137.29    78.5 2134.51    88.3  2131.6
      90 2131.32    98.1 2129.96     105 2130.17   107.9 2130.26   117.7 2132.31
   127.6 2134.82   137.4 2136.56   147.2 2137.72     157 2139.31   166.8 2141.64
   176.6 2144.05   186.4 2146.69   196.2 2149.48
#Mann= 3 , 0 , 0
       0      .1       0      90    .045       0   117.7      .1       0
Bank Sta=90,117.7
XS Rating Curve= 0 ,0
Exp/Cntr=0.3,0.1

Type RM Length L Ch R = 1 ,45007.6 ,540.5,529.7,518.6
XS GIS Cut Line= 3
     1955923.968      395251.593     1956080.218      395352.288
     1956434.385      395428.677
#Sta/Elev= 30
       0 2175.69    39.1 2164.52    58.7 2160.02   107.6 2150.51   156.5 2142.53
   166.3 2140.65   176.1 2137.72   185.9 2134.19   205.5  2127.8   215.3 2124.86
     225 2122.86   234.8 2122.24   244.6 2122.49   283.8 2124.31   293.6 2124.57
   313.2 2124.04   332.8 2123.04   342.6 2121.94   352.4 2119.61   362.1  2116.9
   371.9 2115.77   381.7 2116.27   391.5 2117.79   411.1 2121.41   430.7 2124.16
   450.3 2126.29   489.4 2129.75   499.2 2131.14     509 2133.43   548.2 2143.77
#Mann= 3 , 0 , 0
       0      .1       0   362.1    .045       0   391.5      .1       0
Bank Sta=362.1,391.5
XS Rating Curve= 0 ,0
Exp/Cntr=0.3,0.1

Type RM Length L Ch R = 1 ,44478   ,333.4,336.8,340.3
XS GIS Cut Line= 2
     1956038.551      395959.927     1956570.669      395813.659
#Sta/Elev= 30
       0 2115.64    96.8 2114.09   116.2 2114.06   135.5 2114.21   164.6 2114.98
   174.3 2114.62     184 2111.53   193.6 2105.06   203.3 2099.37     213 2098.36
   220.1 2099.96   222.7 2100.55   232.4 2103.28     242 2104.82   251.7 2105.49
   280.8 2107.14   319.5  2108.6   329.2 2109.06   377.6 2111.75   387.3 2112.43
     397 2113.33   406.6 2114.47   416.3  2115.8     426 2117.28     455 2122.23
   503.4 2129.85   513.1 2131.55   522.8 2133.54   532.5 2135.77   551.8 2140.71
#Mann= 3 , 0 , 0
       0      .1       0   203.3    .045       0   220.1      .1       0
Bank Sta=203.3,220.1
XS Rating Curve= 0 ,0
Exp/Cntr=0.3,0.1

Type RM Length L Ch R = 1 ,44141.2 ,318,335.9,352.7
XS GIS Cut Line= 3
      1955763.51      396074.375     1956109.864      396233.229
     1956646.322      396175.937
#Sta/Elev= 30
       0 2123.41    48.8 2115.21    58.6 2113.85    68.4 2113.09    97.7 2112.04
   146.6 2110.74   234.5 2109.54   351.7 2107.56   430.1 2105.35   439.9 2105.28
   469.3 2105.93   498.8 2106.32   508.6 2106.13   547.8 2103.46   567.4 2101.69
   577.2 2100.54   596.8 2097.53   636.1 2090.67   645.9 2089.53   655.7 2089.54
   665.5 2090.14   802.8 2100.08   812.6 2100.95   822.5  2103.1   832.3 2107.56
   842.1 2113.37   851.9 2119.46   891.1 2144.26   900.9 2150.14   920.6 2161.25
#Mann= 3 , 0 , 0
       0      .1       0   636.1    .045       0   665.5      .1       0
Bank Sta=636.1,665.5
XS Rating Curve= 0 ,0
Exp/Cntr=0.3,0.1

Type RM Length L Ch R = 1 ,43805.3 ,549.1,547,542.9
XS GIS Cut Line= 2
     1955984.864      396204.583     1956601.051      396653.503
#Sta/Elev= 30
       0 2107.97   117.3 2104.66   127.1 2104.33   146.6  2103.1   156.4 2101.99
   195.5 2094.54   205.2  2093.1     215 2092.46     303 2091.16   332.3 2091.44
   410.5 2093.08   459.4 2091.95   488.7    2092   498.5 2090.77     518 2087.33
   527.8 2086.23   537.6 2085.72   557.1 2085.04   566.9 2085.59   576.7 2087.64
   586.4 2091.86   596.2 2096.59     606 2100.55   615.8  2103.9   625.5 2106.67
   635.3 2108.74   645.1 2109.63   713.5 2114.41   752.6 2117.91   762.4 2118.55
#Mann= 3 , 0 , 0
       0      .1       0   537.6    .045       0   566.9      .1       0
Bank Sta=537.6,566.9
XS Rating Curve= 0 ,0
Exp/Cntr=0.3,0.1

Type RM Length L Ch R = 1 ,43258.3 ,442.7,454.4,466
XS GIS Cut Line= 2
     1955728.655      396416.958     1956047.666      396670.864
#Sta/Elev= 30
       0 2101.15     9.7 2102.08    19.4 2102.11    29.1 2101.68    48.5 2100.06
    87.4 2096.09    97.1 2095.22   116.5 2093.63   126.2 2092.49   135.9 2090.81
   174.7 2083.35   184.4 2081.71   203.9 2078.82   213.6 2077.55   223.3 2076.78
     233 2076.51   242.7 2076.54   252.4 2076.89   271.8 2078.78   281.5 2079.96
   291.2 2081.35   300.9 2083.19   310.6 2084.73   320.4 2085.54   330.1 2085.96
   339.8 2086.64   349.5 2087.54   359.2 2088.57   368.9 2089.74   407.7  2094.8
#Mann= 3 , 0 , 0
       0      .1       0   223.3    .045       0   252.4      .1       0
Bank Sta=223.3,252.4
XS Rating Curve= 0 ,0
Exp/Cntr=0.3,0.1

Type RM Length L Ch R = 1 ,42803.8 ,567.2,598.2,629
XS GIS Cut Line= 2
     1955548.534      396781.541      1955807.78      397186.354
#Sta/Elev= 30
       0 2078.28     9.8 2077.55    19.6 2077.14    29.4 2077.12    78.5 2078.11
    88.3 2076.98    98.1 2074.31     1092070.452   117.7 2067.38   127.5 2065.47
   137.4 2066.11   147.2 2068.82   153.7 2070.83     157 2071.85   166.8 2074.54
   215.8 2087.72   225.6 2089.87   235.4 2091.39   245.3 2092.41   255.1 2093.21
   274.7 2094.44   313.9 2096.42   353.2 2098.85   372.8 2100.32   402.2 2102.79
   431.7 2105.37   441.5 2106.36   451.3 2107.53   461.1 2108.91   480.7 2112.05
#Mann= 3 , 0 , 0
       0      .1       0     109    .045       0   153.7      .1       0
Bank Sta=109,153.7
XS Rating Curve= 0 ,0
Exp/Cntr=0.3,0.1

Type RM Length L Ch R = 1 ,42205.7 ,437.3,419.4,401.5
XS GIS Cut Line= 2
      1955179.61      396694.736     1954930.176      396941.562
#Sta/Elev= 27
       0 2066.14     9.8 2063.36    19.5 2062.07    29.2 2062.05      39 2062.27
    48.7 2062.05    58.5 2061.39    68.2 2060.46    87.7 2058.82    97.5  2057.1
     117  2049.5   126.7 2046.93   136.5 2047.43   146.2 2049.64     156 2052.16
   175.5 2056.92     195 2061.92   204.7 2064.56   243.7 2075.44   253.4 2077.57
   263.2 2079.04   272.9 2080.29   282.7 2081.73   302.2 2084.86   321.7 2088.19
   331.4 2089.93   350.9 2093.68
#Mann= 3 , 0 , 0
       0      .1       0     117    .045       0   146.2      .1       0
Bank Sta=117,146.2
XS Rating Curve= 0 ,0
Exp/Cntr=0.3,0.1

Type RM Length L Ch R = 1 ,41786.3 ,617,613.1,609.1
XS GIS Cut Line= 2
      1954706.52      396536.316      1954706.52      396790.222
#Sta/Elev= 28
       0 2056.26     9.8 2051.13    19.5 2047.76    29.3 2046.93    39.1  2047.2
    48.8 2047.52    58.6 2047.81    68.4 2048.02    78.1 2048.14    87.9 2048.12
    97.7 2047.48   107.4 2045.79   117.2 2043.21   126.8 2040.75   136.7 2039.54
   141.8 2040.12   146.5 2040.66   156.2 2043.94     166 2047.86   175.8 2051.24
   185.6 2054.15   195.3 2056.69   205.1 2058.96   214.8 2061.23   224.6  2063.5
   234.4 2065.74   244.1 2067.97   253.9 2070.24
#Mann= 3 , 0 , 0
       0      .1       0   126.8    .045       0   146.5      .1       0
Bank Sta=126.8,146.5
XS Rating Curve= 0 ,0
Exp/Cntr=0.3,0.1

Type RM Length L Ch R = 1 ,41173.2 ,461.1,483.3,505.5
XS GIS Cut Line= 2
      1954079.35       396603.59     1954137.944       396918.26
#Sta/Elev= 23
       0 2051.61     9.7 2049.88    29.1 2046.57      97 2035.37   106.7 2033.68
   116.4 2031.76   123.2 2030.51   126.1 2029.98   135.8 2029.14   145.5 2029.73
   155.2 2031.42   164.9 2033.45   174.6 2035.28   184.3 2036.89   203.7 2039.72
   223.1 2042.34   242.5 2045.07   271.6 2048.61   281.3 2050.51     291 2053.22
   300.7 2056.42   310.4 2060.08   320.1  2064.5
#Mann= 3 , 0 , 0
       0      .1       0   123.2    .045       0   155.2      .1       0
Bank Sta=123.2,155.2
XS Rating Curve= 0 ,0
Exp/Cntr=0.3,0.1

Type RM Length L Ch R = 1 ,40689.9 ,467,458.4,449.7
XS GIS Cut Line= 2
     1953740.808      396614.441     1953528.135      396822.774
#Sta/Elev= 18
       0 2039.74      48 2032.58    57.6 2031.23    76.8 2028.75      96 2026.54
   105.6 2024.98   115.2 2022.64   124.8 2020.01   134.4 2018.36     144 2018.67
   153.22020.576   153.7 2020.68   182.5 2030.51   192.1 2034.09   211.3 2041.51
   220.9 2044.99   249.7  2055.1   297.7 2072.54
#Mann= 3 , 0 , 0
       0      .1       0   115.2    .045       0   153.2      .1       0
Bank Sta=115.2,153.2
XS Rating Curve= 0 ,0
Exp/Cntr=0.3,0.1

Type RM Length L Ch R = 1 ,40231.5 ,731.4,734,735.8
XS GIS Cut Line= 2
     1953445.669      396202.114     1953285.079      396573.208
#Sta/Elev= 28
       0 2058.46     9.6 2056.56    19.2 2054.37    28.9 2051.61      77 2036.38
    96.3 2030.42   105.9 2027.37   115.5 2023.94   125.2 2019.91   134.8 2015.28
   144.4 2010.24   147.12009.256     154 2006.74   163.7 2005.78   173.3 2006.58
   182.9 2007.96   192.6 2009.32   221.4 2013.04   240.7 2015.27   250.3 2016.16
   259.9 2016.88   317.7 2020.96   327.3 2021.92     337 2023.95   346.6 2026.95
   385.1 2039.62   394.7 2042.75   404.4  2045.8
#Mann= 3 , 0 , 0
       0      .1       0   147.1    .045       0   182.9      .1       0
Bank Sta=147.1,182.9
XS Rating Curve= 0 ,0
Exp/Cntr=0.3,0.1

Type RM Length L Ch R = 1 ,39497.5 ,717.2,735.4,753.5
XS GIS Cut Line= 2
     1952783.777      396186.923      1952681.78      396419.128
#Sta/Elev= 29
       0 2011.35     9.8 2010.12    19.5 2008.67    29.3 2006.67      39 2004.15
    48.8 2001.48    58.5 1998.78    68.3 1996.05      78  1993.3    87.8 1990.35
    97.6    1987   105.2 1985.06   107.3 1984.52     117 1983.97   120.2 1984.39
   126.8 1985.26   136.6 1987.54   146.3  1989.9   156.1 1992.05   165.8 1994.19
   175.6 1996.35   185.3 1998.59   195.1 2001.31   204.8 2004.58   214.6 2008.05
   224.4 2011.56   234.1  2015.1   243.9 2018.65   253.6 2022.22
#Mann= 3 , 0 , 0
       0      .1       0   105.2    .045       0   126.8      .1       0
Bank Sta=105.2,126.8
XS Rating Curve= 0 ,0
Exp/Cntr=0.3,0.1

Type RM Length L Ch R = 1 ,38762.1 ,665.6,643.5,621.4
XS GIS Cut Line= 2
     1952330.218      395802.809     1952013.378      395922.166
#Sta/Elev= 29
       0 2000.47      29 1995.66      58  1991.1    67.7 1988.94    77.4 1986.18
    87.1 1983.17    96.7 1979.91   116.1 1973.16   125.8 1970.04   135.4 1967.28
   145.1 1964.94   154.8 1963.48   155.41963.465   164.4 1963.25   174.1 1964.54
   183.1 1967.24   193.5 1970.47   203.2 1973.33   212.8 1976.34   222.5  1978.9
   232.2 1980.62   241.8 1981.91   251.5 1983.35   280.5 1987.91   299.9 1990.71
   309.6 1992.24   319.2 1994.15   328.9 1996.36   338.6 1998.39
#Mann= 3 , 0 , 0
       0      .1       0   155.4    .045       0   183.1      .1       0
Bank Sta=155.4,183.1
XS Rating Curve= 0 ,0
Exp/Cntr=0.3,0.1

Type RM Length L Ch R = 1 ,38118.6 ,731.7,727.4,723
XS GIS Cut Line= 2
     1951796.364      395268.955      1951731.26      395525.031
#Sta/Elev= 30
       0 1971.53     9.8 1970.75    19.6    1970    29.4 1969.05    39.1 1967.68
    48.9 1965.62    58.7 1962.59    68.5 1958.79    78.3 1954.76    88.1 1950.76
    97.9 1946.78   107.6 1942.78   117.4 1938.77   127.2 1934.36     137 1930.08
   138.2 1929.84   146.8 1928.12   153.2 1929.05   156.6 1929.54   166.4 1934.48
   176.2  1940.8   185.9 1946.28   195.7 1950.97   205.5  1955.3   215.3 1959.47
   225.1 1963.49   234.9 1967.06   244.6 1969.67   254.4  1971.4   264.2 1972.76
#Mann= 3 , 0 , 0
       0      .1       0     137    .045       0   156.6     .06       0
Bank Sta=137,156.6
XS Rating Curve= 0 ,0
Exp/Cntr=0.3,0.1

Type RM Length L Ch R = 1 ,37391.2 ,634.8,639,643
XS GIS Cut Line= 2
     1951047.666      395286.316     1951019.454      395750.725
#Sta/Elev= 30
       0 1952.54    38.8 1942.39    48.5 1939.98    58.2 1937.96    96.9 1931.97
   106.6 1930.12   116.3    1928     126 1926.62   135.7 1926.75   145.4 1927.84
   155.1  1928.8   164.8 1929.39   174.5 1929.66   193.9 1929.62   222.9 1929.27
   232.6  1929.4   290.8 1932.09   300.5 1932.82   310.2 1935.04   319.9 1939.04
   329.6 1943.83     349 1953.65   358.6 1958.94   368.3 1965.07     378 1971.64
   387.7 1977.15   397.4 1981.18   407.1 1984.36   416.8  1987.1   465.3  1999.6
#Mann= 3 , 0 , 0
       0      .1       0   116.3    .045       0   145.4     .06       0
Bank Sta=116.3,145.4
XS Rating Curve= 0 ,0
Exp/Cntr=0.3,0.1

Type RM Length L Ch R = 1 ,36752.2 ,499.3,495.4,490.8
XS GIS Cut Line= 2
     1950455.218      395162.618     1950390.114      395446.906
#Sta/Elev= 21
       0 1932.44     9.7 1932.11    19.4 1931.21    29.2 1929.74    58.3 1924.22
    77.8 1920.92   116.7 1913.34   126.4 1911.57   145.8  1908.5   155.6 1907.29
   165.3 1906.99     175 1907.69   184.7 1909.39   194.4 1911.18   204.2  1912.6
   213.9 1913.74   223.6 1915.03   233.3 1916.92     243 1919.21   252.8 1921.74
   291.6 1932.37
#Mann= 3 , 0 , 0
       0      .1       0   145.8    .045       0   184.7     .06       0
Bank Sta=145.8,184.7
XS Rating Curve= 0 ,0
Exp/Cntr=0.3,0.1

Type RM Length L Ch R = 1 ,36256.8 ,210.1,210,210.7
XS GIS Cut Line= 2
     1949953.916      395025.899     1949925.704      395462.097
#Sta/Elev= 28
       0 1915.63     9.7 1913.65    19.4 1912.12    48.6 1907.72    58.3 1906.64
      68 1906.02    77.7 1906.06    87.4 1907.08    97.1 1908.65   106.8 1909.43
   116.6 1908.78     136 1905.96   155.4 1902.91   165.1 1902.22   174.8 1902.82
   183.1 1903.74   184.6 1903.91   194.3 1904.58     204 1904.75   301.1 1905.25
   359.4 1905.33   369.1 1905.52   378.8  1906.5   388.5  1908.8   398.3 1912.12
   417.7 1919.38   427.4 1922.75   437.1 1925.49
#Mann= 3 , 0 , 0
       0      .1       0   155.4    .045       0   183.1      .1       0
#XS Ineff= 2 , 0
          106.34 1909.42
Permanent Ineff=
       F       F
Bank Sta=155.4,183.1
XS Rating Curve= 0 ,0
Exp/Cntr=0.3,0.1

Type RM Length L Ch R = 1 ,36046.8 ,43.4,43.4,43.4
XS GIS Cut Line= 3
     1949748.295      394949.944     1949730.934      395251.593
     1949600.726       395514.18
#Sta/Elev= 30
       0 1907.96    19.5 1907.12    58.5 1904.87      78 1903.99    97.5 1903.32
   146.2 1902.53   204.7  1901.1   224.2  1900.1   243.7 1898.51   253.4 1896.75
   263.2 1896.26   272.9  1897.8   282.7 1899.93   292.4 1900.63   331.5 1900.76
   360.8 1900.06   370.5 1900.13   380.3  1900.5   399.8  1901.9   409.6 1902.43
   438.9 1903.39     478 1905.12   497.6 1905.68   517.1 1906.04   526.9  1906.6
   536.6 1907.87   546.4 1909.83   556.2  1911.3   585.5 1914.26   595.2 1915.11
#Mann= 3 , 0 , 0
       0      .1       0   243.7    .045       0   272.9      .1       0
Bank Sta=243.7,272.9
XS Rating Curve= 0 ,0
Exp/Cntr=0.3,0.1

Type RM Length L Ch R = 1 ,36003.4 ,241.6,242.7,243.8
XS GIS Cut Line= 3
     1949704.892      394949.944     1949687.531      395251.593
     1949557.323       395514.18
#Sta/Elev= 30
       0 1906.73    19.5  1906.7    29.2 1906.36    58.5 1904.86    87.7 1903.72
   107.2 1903.33   126.7 1903.15   185.2 1901.29   204.7 1901.21   224.2 1902.33
   233.9 1902.12   243.7 1899.71   253.4  1896.6   263.2  1895.9   272.9 1897.92
   282.7 1900.55   292.4 1901.58   302.2 1901.34   321.7 1900.37   331.5 1900.05
     351 1900.11   360.8 1900.67   370.5 1901.43   380.3 1901.91   419.4  1903.1
     478  1906.1   507.3 1907.19   517.1 1907.77   536.6 1909.35   595.2 1914.69
#Mann= 3 , 0 , 0
       0      .1       0   243.7    .045       0   272.9      .1       0
#XS Ineff= 2 , 0
           223.1 1902.44
Permanent Ineff=
       F       F
Bank Sta=243.7,272.9
XS Rating Curve= 0 ,0
Exp/Cntr=0.3,0.1

Type RM Length L Ch R = 1 ,35760.7 ,537.8,528.9,519.5
XS GIS Cut Line= 2
     1949476.485      394973.816     1949428.742      395420.864
#Sta/Elev= 21
       0 1900.97    58.6  1898.8      88 1897.86    97.7 1897.66   107.5 1897.59
   136.8 1897.57   146.6 1897.09   156.4 1895.33   159.7 1894.58   166.2 1893.11
   175.9 1892.35   185.7 1893.64   195.5 1895.48   205.2 1895.76     215 1895.13
   224.8 1895.02   244.3 1895.78   263.9 1896.42   283.4 1896.87   371.4  1898.1
   449.6 1898.96
#Mann= 3 , 0 , 0
       0      .1       0   159.7    .045       0   185.7     .08       0
Bank Sta=159.7,185.7
XS Rating Curve= 0 ,0
Exp/Cntr=0.3,0.1

Type RM Length L Ch R = 1 ,35231.8 ,539,555.5,571.8
XS GIS Cut Line= 2
     1948955.652      395138.746     1949059.819      395598.816
#Sta/Elev= 30
       0  1893.3    39.3 1893.38      59 1893.09    78.6  1892.6    98.3 1892.54
   117.9 1892.78   127.8 1892.75   137.6 1892.47   147.4 1891.69   157.2 1890.37
   167.1 1888.59   176.9 1886.18   196.6 1879.44   206.4 1877.66   216.2 1877.58
     226 1878.84   255.5 1884.33   265.3 1885.87   275.2 1886.92     285 1887.39
   314.5 1887.83     344 1887.84   383.3  1888.1   402.9 1887.92   422.6 1887.52
   432.4 1887.94   442.2 1889.94   452.1 1893.11   461.9 1896.85   471.7 1901.24
#Mann= 3 , 0 , 0
       0      .1       0   196.6    .045       0     226      .1       0
Bank Sta=196.6,226
XS Rating Curve= 0 ,0
Exp/Cntr=0.3,0.1

Type RM Length L Ch R = 1 ,34676.3 ,785.7,791.7,797.7
XS GIS Cut Line= 2
     1948543.326      395273.295     1948404.437      395533.711
#Sta/Elev= 25
       0 1882.64    49.2 1883.13    78.7 1883.26    88.5 1883.48    98.4 1883.88
   108.2 1883.89   118.1  1883.1   127.9  1881.6   137.7 1879.66   148.91876.593
   157.4 1874.06   167.2 1872.75   177.1 1873.18   186.71874.806   196.8 1876.83
   206.6  1879.6   216.4  1884.4   226.3 1890.59   236.1  1897.8     246 1905.55
   255.8 1912.94   265.6 1919.43   275.5 1925.61   285.3 1931.49   295.1 1936.44
#Mann= 3 , 0 , 0
       0      .1       0   148.9    .045       0   186.7      .1       0
Bank Sta=148.9,186.7
XS Rating Curve= 0 ,0
Exp/Cntr=0.3,0.1

Type RM Length L Ch R = 1 ,33884.6 ,911,888.9,866.7
XS GIS Cut Line= 2
     1948382.735      394509.406     1947961.728      394939.093
#Sta/Elev= 30
       0 1955.36     9.7  1950.2    19.4 1944.66    29.1 1939.73    38.8 1935.51
    48.5 1931.73    58.2 1928.96    67.9 1926.88    77.6 1924.44    87.3 1920.29
   135.8 1897.15   155.2 1888.27   164.9 1884.29   174.6  1881.2   184.4 1879.08
     194 1877.33   252.3 1868.43   281.4 1863.81   291.1 1862.62   300.8 1862.06
   310.5 1862.13   329.9 1862.94     359 1864.58   407.5 1868.28   417.2 1868.81
   426.9 1869.14     456  1869.4   494.8 1869.49   543.4 1870.36   601.6 1871.12
#Mann= 3 , 0 , 0
       0      .1       0   291.1    .045       0   329.9      .1       0
Bank Sta=291.1,329.9
XS Rating Curve= 0 ,0
Exp/Cntr=0.3,0.1

Type RM Length L Ch R = 1 ,32995.7 ,725.2,726.1,726.9
XS GIS Cut Line= 3
     1947393.152      394309.753     1947397.492      394492.045
      1947514.68      394999.857
#Sta/Elev= 30
       0 1939.57     9.6 1934.91    19.2 1930.56    57.6 1914.87    86.4 1901.85
      96 1898.06   115.2 1891.25   124.8 1887.61   134.4 1883.42   163.2  1870.2
   182.3 1862.64     202 1854.26   211.8 1851.91   221.7 1851.68   241.3 1853.44
     261 1854.88   280.7 1855.76   290.5 1855.95   300.3 1855.88   329.8 1854.91
   349.5 1854.61   369.2 1854.77   388.8 1855.23   447.8 1857.85     497 1859.53
   624.8 1863.71   644.5 1864.27     674 1864.76   683.8 1865.16   703.5 1866.97
#Mann= 3 , 0 , 0
       0      .1       0     202    .045       0   241.3      .1       0
Bank Sta=202,241.3
XS Rating Curve= 0 ,0
Exp/Cntr=0.3,0.1

Type RM Length L Ch R = 1 ,32269.7 ,471.5,453,434.5
XS GIS Cut Line= 2
      1946683.71      394571.908     1946793.326      395145.691
#Sta/Elev= 30
       0 1862.29    48.7 1856.14    77.9 1851.58    87.6 1850.77    97.4 1850.64
   107.1 1850.24   136.3 1846.83   155.8 1845.17   165.5 1844.53   175.2 1844.16
     185 1844.43   194.7 1845.27   214.2  1846.9   223.9 1847.55   233.7 1847.89
   272.6 1847.64   311.6 1846.38     331 1846.01   350.5 1845.87     370 1846.04
   389.4  1846.5   408.9 1847.33   428.4  1848.4   447.9  1849.1   457.6 1849.18
   486.8 1848.89   525.7 1848.79   545.2 1848.96   574.4 1848.95   584.2 1849.24
#Mann= 3 , 0 , 0
       0      .1       0   155.8    .045       0   194.7      .1       0
Bank Sta=155.8,194.7
XS Rating Curve= 0 ,0
Exp/Cntr=0.3,0.1

Type RM Length L Ch R = 1 ,31816.7 ,520.8,510.2,499.7
XS GIS Cut Line= 2
     1946173.968      394825.378     1946798.968      395216.003
#Sta/Elev= 30
       0  1883.7     9.8 1879.37    19.6 1875.74    29.5 1872.41    39.3 1869.64
    68.8 1862.43    98.3 1855.93   137.6 1844.91   147.4  1842.4   157.2 1840.65
   167.1 1839.87   176.9  1839.8   196.5 1840.43   235.8 1842.12   255.5 1842.51
   294.8  1844.3   314.5 1844.06     344 1842.73   363.6 1842.28   461.9  1841.9
   471.7 1841.25   501.2 1837.02   520.8 1835.16   530.7 1835.38   540.5 1836.97
   560.1 1841.54     570 1842.51   628.9 1844.36   668.2 1846.05     737 1851.58
#Mann= 3 , 0 , 0
       0      .1       0   157.2    .045       0   196.5      .1       0
#XS Ineff= 2 , 0
                          295.21         1844.55
Permanent Ineff=
       F       F
Bank Sta=157.2,196.5
XS Rating Curve= 0 ,0
Exp/Cntr=0.3,0.1
